--- Barrenshe Creek.prj (project) ---

Proj Title=Barrenshe Creek
Current Plan=p01
Default Exp/Contr=0,0
English Units
Geom File=g01
Flow File=f01
Plan File=p01
BEGIN DESCRIPTION:
END DESCRIPTION:
DSS Export Rating Curves= 0
DSS Export Rating Curve Sorted= 0
DSS Export Volume Flow Curves= 0
DXF OffsetX= 0
DXF OffsetY= 0
DXF ScaleX= 0
DXF ScaleY= 0

--- Barrenshe Creek.p01 (plan) ---

Plan Title=Floodplain
Program Version=4.00
Geom File=g01
Flow File=f01
K Sum by GR=0
Std Step Tol=0.01
Critical Tol=0.01
Num of Std Step Trials=20
Max Error Tol=0.3
Flow Tol Ratio=0.001
Split Flow NTrial=30
Split Flow Tol=0.02
Split Flow Ratio=0.02
Log Output Level=0
Friction Slope Method=1
Unsteady Friction Slope Method=2
Unsteady Bridges Friction Slope Method=1
Global Log Level=0
CheckData=False
Run HTab=0
Run UNet=0
Run PostProcess=0
UNET Theta=0
UNET Theta Warmup=0
UNET ZTol=0
UNET ZSATol=0
UNET MxIter=0
UNET MaxInSteps=0
UNET DtIC=0
UNET DtMin=0
UNET MaxCRTS=0
UNET WFStab=0
UNET SFStab=0
UNET WFX=0
UNET SFX=0
UNET DSS MLevel=0
UNET DZMax Abort=0
UNET Convert EG Bridges=0
UNET Use Existing IB Tables=0
UNET Froude Limit=0
UNET Froude Power=0
Write IC File=0
Echo Input=False
Echo Output=False
Write Detailed=0

--- Barrenshe Creek.f01 (steady flow) ---

Flow Title=NFF Regression Equation
Program Version=4.00
Number of Profiles=1
Profile Names=P100yr
River Rch & RM=Barrenshe Creek,Main      ,19693.4
626.1812
River Rch & RM=Barrenshe Creek,Main      ,17933.8
660.3924
River Rch & RM=Barrenshe Creek,Main      ,17627
774.4855
River Rch & RM=Barrenshe Creek,Main      ,17329.4
834.8209
River Rch & RM=Barrenshe Creek,Main      ,15214.8
885.0308
River Rch & RM=Barrenshe Creek,Main      ,14923.1
1024.913
River Rch & RM=Barrenshe Creek,Main      ,12839.3
1092.986
River Rch & RM=Barrenshe Creek,Main      ,12561.7
1262.231
River Rch & RM=Barrenshe Creek,Main      ,12192.2
1272.774
River Rch & RM=Barrenshe Creek,Main      ,9567.7
1407.818
River Rch & RM=Barrenshe Creek,Main      ,9269.1
1750.220
River Rch & RM=Barrenshe Creek,Main      ,6569.3
1816.530
River Rch & RM=Barrenshe Creek,Main      ,6259.7
2243.922
River Rch & RM=Barrenshe Creek,Main      ,285
2456.917
Boundary for River Rch & Prof#=Barrenshe Creek,Main      ,1
Up Type=0
Dn Type=3
Dn Slope=0.022494

--- Barrenshe Creek.g01 (geometry) ---

Geom Title=USGS 10m DEM
Program Version=4.00

River Reach=Barrenshe Creek ,Main
Reach XY= 30
     1781337.093      124261.178     1781192.446      124082.809
      1780892.28      124012.578     1780669.953      123720.634
     1779437.953      123314.151     1778443.915      122385.909
     1778393.842      122155.704     1778033.181      121610.792
     1777255.727      121367.348     1776927.719      121403.112
     1776748.987      121633.643       1774615.3       121679.09
     1773800.684      121811.024     1773106.353      122041.864
     1772718.903      122270.893     1772475.961      122139.854
      1772036.86      122272.821     1771054.139      122160.881
     1770627.407      122037.809     1770211.807      121826.299
     1769142.442      120776.027     1768648.978      119928.269
     1768655.917      119486.913     1768409.996      118664.508
     1767703.694      117904.348     1766945.227      117631.177
     1766632.663      117755.504     1766319.605      117725.573
     1766089.059      117610.704     1765967.625      117409.851

Type RM Length L Ch R = 1 ,19693.4 ,273.6,263.4,253.2
XS GIS Cut Line= 3
     1781717.789      123944.471     1781333.426      124251.875
     1780920.286      124581.478
#Sta/Elev= 30
      10  1865.5    40.2 1846.23    60.3 1835.99   150.7 1804.67   210.9 1777.99
     231 1766.05   271.2  1734.5   291.3 1720.79   321.4 1703.84   371.6 1680.78
   411.8 1664.73   431.9 1661.68   489.6  1656.4   502.1 1656.19   514.6 1656.96
   532.1 1661.93     562 1673.37   581.9 1678.53   621.8 1685.43   651.7 1689.08
   741.5 1707.37   851.2 1722.93   881.1 1728.48     901  1734.2   950.9 1754.53
   970.8 1765.69   990.8 1773.82  1000.7 1779.87  1010.7 1788.45  1020.7 1794.77
#Mann= 3 , 0 , 0
       0     .08       0   489.6    .045       0   514.6     .08       0
Bank Sta=489.6,514.6
XS Rating Curve= 0 ,0
Exp/Cntr=0.3,0.1

Type RM Length L Ch R = 1 ,19430   ,334.3,335.5,336.7
XS GIS Cut Line= 4
     1781388.498      123712.939     1781234.143      123934.181
     1781074.643       124212.02     1780873.982      124505.294
#Sta/Elev= 30
      10 1826.13      30 1814.91      40 1810.81    79.9 1802.61   159.9 1771.03
   179.8 1759.66   289.8 1692.04   349.9 1663.86   369.9  1656.2   417.4 1646.78
   429.9 1645.88   442.4 1646.73     480 1649.71     500 1652.37   520.1 1658.27
   530.1 1662.19   550.1 1673.04   570.1 1687.38   590.1 1705.05   629.6 1744.24
   659.2 1771.35   669.1 1779.59     679 1786.12   688.8 1789.88   708.6 1791.94
   797.4 1796.66   836.9 1803.36   896.1 1809.28   935.6  1818.9   945.5 1822.48
#Mann= 3 , 0 , 0
       0     .08       0   417.4    .045       0   442.4     .08       0
Bank Sta=417.4,442.4
XS Rating Curve= 0 ,0
Exp/Cntr=0.3,0.1

Type RM Length L Ch R = 1 ,19094.5 ,269,273.2,277.1
XS GIS Cut Line= 3
     1781185.542      123535.078     1780857.049      123976.188
     1780585.853      124335.504
#Sta/Elev= 30
      10 1885.19      20 1883.56      30 1878.71      50 1864.02      90 1830.35
     120 1807.82     150 1786.28     200 1753.04     270 1709.17     320 1681.37
     360 1662.49     380 1656.32     450 1638.83   487.5 1635.09     500 1634.61
   512.5 1634.78     560 1636.91     570 1638.04     580 1641.55     590  1648.8
     600 1657.56     640 1694.22     710 1764.49   760.1 1812.94   780.1 1830.67
   800.1  1846.3   820.1  1859.3   850.1 1875.19   940.1 1926.86  1000.2 1957.78
#Mann= 3 , 0 , 0
       0     .08       0   487.5    .045       0   512.5     .08       0
Bank Sta=487.5,512.5
XS Rating Curve= 0 ,0
Exp/Cntr=0.3,0.1

Type RM Length L Ch R = 1 ,18821.4 ,258.7,255.1,249.4
XS GIS Cut Line= 4
     1780925.433      123352.777     1780796.804      123630.616
     1780621.869      123857.003     1780452.078      124191.439
#Sta/Elev= 30
     9.9 1826.38    39.5 1817.42    59.3 1807.77    88.9 1790.07   148.1 1751.62
   187.7  1727.1   217.3 1710.86   246.9 1696.56   286.4 1679.01   335.8 1661.46
   385.1 1642.02   414.7 1632.81   431.8 1630.73   444.3 1630.57   456.8 1630.65
   483.7  1631.3   493.6  1633.7   533.1 1648.64   562.7 1664.49   582.4 1676.56
   641.6 1715.13   710.7 1755.64   750.2 1780.83   769.9 1796.72   809.4  1835.8
   819.3 1844.89   829.2 1853.05     839 1859.84   898.2 1888.73   967.3 1915.75
#Mann= 3 , 0 , 0
       0     .08       0   431.8    .045       0   456.8     .08       0
Bank Sta=431.8,456.8
XS Rating Curve= 0 ,0
Exp/Cntr=0.3,0.1

Type RM Length L Ch R = 1 ,18566.3 ,637,632.5,627.9
XS GIS Cut Line= 3
     1780726.299        123189.8     1780493.824      123633.117
     1780268.331      124079.928
#Sta/Elev= 30
      10 1702.76    50.1 1699.13   110.1 1687.86   140.2 1683.44   170.2 1680.74
   210.2 1678.61   230.3 1676.67   250.3 1673.53   270.3 1669.13   290.3 1662.97
   340.4  1643.2   360.4 1639.62   380.4 1637.88   430.5 1637.36   508.1 1627.96
   520.6 1626.53   533.1 1627.21   540.6 1628.98   560.6 1638.94   590.7 1651.68
   610.7 1662.33   690.8 1708.01   750.8 1744.51   810.9 1783.38   880.9 1826.46
     901 1837.93     921  1847.7     931 1851.46     971 1864.59  1001.1 1873.21
#Mann= 3 , 0 , 0
       0     .08       0   508.1    .045       0   533.1     .08       0
Bank Sta=508.1,533.1
XS Rating Curve= 0 ,0
Exp/Cntr=0.3,0.1

Type RM Length L Ch R = 1 ,17933.8 ,309.3,306.9,304.5
XS GIS Cut Line= 4
     1780091.427      122990.705      1779972.42      123217.186
     1779886.156       123514.71     1779729.782      123927.745
#Sta/Elev= 30
     9.8 1777.39    49.2 1756.58    98.4 1733.36   137.8 1719.73   206.6 1681.27
   236.2 1667.77   255.8 1661.48   295.8 1652.81   315.8 1646.94   365.8 1624.78
   375.8  1621.2   385.8 1620.28   395.7 1621.79   405.7 1621.54   425.7 1614.55
   473.2  1612.7   485.7 1612.13   498.2 1613.18   505.7 1615.24   525.6 1626.93
   595.7    1659   635.9 1683.37     666 1698.52   736.3 1737.23   826.6 1789.18
   896.9 1832.04     937 1857.74   957.1  1872.2   987.2 1895.74  1007.3 1909.95
#Mann= 3 , 0 , 0
     9.8     .08       0   473.2    .045       0   498.2     .08       0
#XS Ineff= 2 , 0
          457.03  1629.3
Permanent Ineff=
       F       F
Bank Sta=473.2,498.2
XS Rating Curve= 0 ,0
Exp/Cntr=0.3,0.1

Type RM Length L Ch R = 1 ,17627   ,276.3,297.5,318.8
XS GIS Cut Line= 4
     1779839.804      122874.277     1779639.142      123244.729
     1779587.691      123501.987     1779582.546      123841.568
#Sta/Elev= 30
      10 1857.15    40.1 1856.12    60.2 1854.11    70.2 1851.02    80.2 1846.35
   100.3 1832.69   150.5 1794.65   210.7 1752.53   270.8 1707.37   290.9 1693.73
   300.9 1688.29   401.2 1639.77   451.6 1617.28   461.7 1613.98   471.8 1612.84
   491.9 1612.47   519.8 1606.48   532.3 1605.02   542.4 1605.91   544.8 1606.92
   552.5 1610.18   572.7 1620.68   633.2 1646.06   693.6 1675.84   783.5 1732.13
   813.5    1750   933.4 1812.81   953.4 1823.94   983.3  1842.4  1023.3 1868.88
#Mann= 3 , 0 , 0
       0     .08       0   519.8    .045       0   544.8     .08       0
Bank Sta=519.8,544.8
XS Rating Curve= 0 ,0
Exp/Cntr=0.3,0.1

Type RM Length L Ch R = 1 ,17329.4 ,346.9,339.9,332.9
XS GIS Cut Line= 4
     1779747.191      122853.696     1779493.345      123139.724
     1779304.092      123273.962     1778987.806      123561.688
#Sta/Elev= 30
    10.1 1876.08    30.2 1861.83    70.4  1830.9   110.7  1804.9     151 1777.92
   231.5 1722.01   281.8 1688.66   301.9 1676.62     443 1605.83     453 1603.39
   473.2 1604.57   483.3 1604.36   493.4 1603.39   531.3 1597.08   543.8 1596.63
   556.3 1598.11   594.3 1607.24   614.5 1612.84   634.3  1616.5     694 1623.65
   793.4 1632.76   823.3 1637.03   843.2 1641.16   853.1    1644     863  1647.6
   952.5 1681.19   972.4 1689.98   982.4 1693.66  1032.1  1710.1    1042 1714.16
#Mann= 3 , 0 , 0
       0     .08       0   531.3    .045       0   556.3     .08       0
Bank Sta=531.3,556.3
XS Rating Curve= 0 ,0
Exp/Cntr=0.3,0.1

Type RM Length L Ch R = 1 ,16989.5 ,286.4,282.2,277.5
XS GIS Cut Line= 4
     1779438.481      122632.454     1779232.674      122910.293
     1779047.449      123110.954     1778821.061      123409.374
#Sta/Elev= 30
     9.9 1779.79    39.5 1776.38    59.3 1768.38   187.7 1702.89   286.5 1650.29
   306.2 1641.12   355.9 1623.52   416.6 1599.52   426.7 1597.05   436.8 1597.09
   467.1  1603.5   477.2 1603.06   495.1 1594.83   507.6 1591.19   520.1 1593.31
   568.3 1613.81   588.5 1624.65   648.4 1660.87     678 1677.36   697.7 1686.11
   707.6 1688.72   717.4 1689.05   756.8 1683.92     816 1681.18   845.6 1681.94
   894.8 1685.87   924.4 1686.22   934.3 1685.72   983.6 1678.38   993.4 1679.53
#Mann= 3 , 0 , 0
       0      .1       0   495.1    .045       0   520.1      .1       0
Bank Sta=495.1,520.1
XS Rating Curve= 0 ,0
Exp/Cntr=0.3,0.1

Type RM Length L Ch R = 1 ,16707.3 ,460.4,468.4,476.9
XS GIS Cut Line= 3
     1779183.418      122436.776     1778904.589      122852.389
      1778633.87      123273.493
#Sta/Elev= 30
      10 1731.76    60.1 1717.36   150.1 1686.92   180.2 1681.31   200.2 1675.38
   240.2 1655.44   280.3 1631.68   320.3 1613.59   340.3 1606.16   410.4 1592.42
   420.4 1591.38   450.4 1592.44   460.4 1591.77     488 1585.68   500.5 1583.62
   510.5 1584.25     513 1585.37   520.5 1588.72   550.5 1608.82   690.7 1689.92
   750.8 1726.25   780.8 1745.29   850.9 1794.08   870.9 1806.15     891 1815.13
     901 1817.58     931 1821.87     951 1826.37   971.1 1832.33  1001.1 1843.27
#Mann= 3 , 0 , 0
       0      .1       0     488    .045       0     513      .1       0
Bank Sta=488,513
XS Rating Curve= 0 ,0
Exp/Cntr=0.3,0.1

Type RM Length L Ch R = 1 ,16238.9 ,379.9,385.8,391.6
XS GIS Cut Line= 4
     1778979.084      122225.399     1778691.506      122428.911
     1778461.003        122619.9     1778253.616      122873.689
#Sta/Elev= 30
    10.1 1789.06    30.2 1772.99    60.4 1750.99    80.5 1738.41   140.9 1703.98
   181.2 1682.06   221.4 1661.83   261.7 1643.46     302 1627.06   342.2 1612.38
   362.3 1605.97   382.2 1600.47   452.1 1582.55   462.1 1581.47     482 1582.69
     492 1581.02   499.5 1578.65     502 1577.87     512 1576.83   524.5 1578.56
   541.9 1582.81   581.8 1589.35   601.8 1594.48   621.7 1601.67   651.7  1615.1
   671.5 1621.48     741 1641.48   810.6 1660.62   949.6 1712.49   979.4 1722.39
#Mann= 3 , 0 , 0
       0      .1       0   499.5    .045       0   524.5      .1       0
Bank Sta=499.5,524.5
XS Rating Curve= 0 ,0
Exp/Cntr=0.3,0.1

Type RM Length L Ch R = 1 ,15853.1 ,278,278.5,279
XS GIS Cut Line= 3
     1778856.151      121997.541     1778432.568      122188.667
      1777970.36      122442.083
#Sta/Elev= 30
    10.1 1759.33    50.5 1745.57    90.9 1729.77   151.5 1703.58   222.3  1670.2
   262.7 1653.57   313.2 1634.55   444.5 1587.14   464.7  1579.2   474.7 1574.69
   484.6 1571.47   494.5  1570.5     507 1570.55   534.3 1570.73   544.3  1571.6
   554.2 1574.88   574.1 1584.77   613.9 1606.05   633.8 1617.47   653.7 1629.73
   683.5 1648.81   753.1 1694.77     783 1714.12   812.8  1732.9   842.6 1750.33
   882.4  1771.5   942.1 1801.26     952 1805.89   971.9 1814.43   991.8 1821.76
#Mann= 3 , 0 , 0
    10.1     .08       0   484.6    .045       0     507     .08       0
Bank Sta=484.6,507
XS Rating Curve= 0 ,0
Exp/Cntr=0.3,0.1

Type RM Length L Ch R = 1 ,15574.5 ,368.5,359.7,348.1
XS GIS Cut Line= 3
     1778700.551      121740.246     1778256.528      121971.219
     1777812.817      122202.772
#Sta/Elev= 30
      10 1824.95      40 1810.96    60.1 1798.79   100.1 1772.07   160.2 1727.32
   170.2 1720.94   190.2 1709.61   290.3 1661.81   340.3 1636.21   370.4 1618.94
   470.5 1575.82   490.5 1565.15     498 1563.08   510.5 1561.98     523 1562.59
   570.6 1564.97   580.6 1566.26   630.6 1578.67   700.7 1596.99   730.7 1605.98
   760.8 1617.74   790.8 1631.57   800.8 1636.77   810.8 1642.98   830.8  1658.5
   850.9 1676.44   880.9  1705.9   920.9 1740.08     971 1784.92    1001 1808.67
#Mann= 3 , 0 , 0
      10     .08       0     498    .045       0     523     .08       0
#XS Ineff= 2 , 0
                          542.24         1593.93
Permanent Ineff=
       F       F
Bank Sta=498,523
XS Rating Curve= 0 ,0
Exp/Cntr=0.3,0.1

Type RM Length L Ch R = 1 ,15214.8 ,309.8,291.7,276.5
XS GIS Cut Line= 4
     1778357.996      121371.889      1778164.17      121594.888
     1777941.238      121788.647     1777750.867      122081.922
#Sta/Elev= 30
     9.8 1664.96    88.6 1665.91   177.3 1660.44     197 1657.17   216.7  1649.9
   295.5  1615.9     325 1599.81   344.7 1588.24   364.4 1576.25   393.9 1556.39
   401.1 1554.92   413.6 1554.26   426.1 1554.65   561.3 1558.73   571.1 1560.36
     581 1564.25   640.8 1600.24   670.7 1617.13   710.7 1637.69   760.7 1660.22
   780.6  1670.2   810.6 1688.05   830.6 1702.36   840.6 1710.68   850.6  1720.1
   860.6 1730.68   890.5 1765.15   910.5 1785.76   930.5 1801.85   940.5 1807.64
#Mann= 3 , 0 , 0
     9.8     .08       0   401.1    .045       0   426.1     .08       0
#XS Ineff= 2 , 0
                          478.33         1575.35
Permanent Ineff=
       F       F
Bank Sta=401.1,426.1
XS Rating Curve= 0 ,0
Exp/Cntr=0.3,0.1

Type RM Length L Ch R = 1 ,14923.1 ,310.6,313.2,315.8
XS GIS Cut Line= 3
     1777914.614      121026.753     1777838.074      121522.814
     1777760.259       122030.06
#Sta/Elev= 30
      10 1746.79   100.4  1729.9   150.6 1716.84   170.7 1710.47   180.7 1705.27
   200.8 1690.39   220.8 1673.58   240.9 1654.22     251 1645.65     261  1639.1
   291.1 1623.22   321.2 1609.69   391.5 1582.88   411.6 1576.48   451.7 1566.99
   489.4 1550.57   491.9 1549.58   501.9 1548.58   514.4 1551.23   532.1 1555.76
   542.2  1556.5   662.9 1553.65     673 1555.02   683.1  1558.7   823.9 1642.53
   914.5 1699.29   954.7 1721.74   984.9 1743.09     995 1751.11  1015.1 1769.11
#Mann= 3 , 0 , 0
       0     .08       0   489.4    .045       0   514.4     .08       0
Bank Sta=489.4,514.4
XS Rating Curve= 0 ,0
Exp/Cntr=0.3,0.1

Type RM Length L Ch R = 1 ,14609.9 ,312.7,307.3,301.8
XS GIS Cut Line= 4
     1777677.833      120983.115     1777554.598      121381.428
     1777499.582       121601.49     1777488.579      121922.781
#Sta/Elev= 30
     9.9 1846.65    49.6 1828.71    69.5 1816.78    89.3 1802.53     139 1761.06
   188.6 1712.95   218.4 1685.91   238.3 1670.14   258.1 1657.35   287.9 1642.65
   327.6 1626.87   367.3 1614.36   416.9 1602.47   436.7 1595.64   466.3 1580.11
   522.8 1545.71   535.3 1543.36   547.8 1545.39   574.7 1550.82   594.5 1552.55
   614.2 1552.06   643.8 1547.61   653.8  1548.1   663.9 1551.19   714.1 1572.07
   744.2 1587.89   794.5 1620.82   864.8 1668.11     915  1705.3   965.3 1733.02
#Mann= 3 , 0 , 0
       0      .1       0   522.8    .045       0   547.8     .08       0
Bank Sta=522.8,547.8
XS Rating Curve= 0 ,0
Exp/Cntr=0.3,0.1

Type RM Length L Ch R = 1 ,14302.6 ,241.3,234.5,227.9
XS GIS Cut Line= 3
     1777277.512      120893.389      1777249.47      121351.287
     1777220.915      121922.421
#Sta/Elev= 30
      10 1680.72    79.8  1681.1    99.7 1683.33   149.6 1692.13   169.5 1693.75
   209.4 1692.85   219.4 1691.58   229.4 1688.85   249.3 1679.19   269.3 1665.31
   299.2 1642.44   319.1 1630.54   349.1 1617.86   398.9 1599.47   408.9 1593.34
   428.8 1574.84   438.8 1564.34   458.8 1541.17   466.3 1536.22   468.8 1534.57
   478.8    1534   491.3 1535.25   569.1 1544.72   609.2  1545.5   659.4 1543.58
   669.4 1544.77   679.5 1548.14   749.7 1579.88   880.1 1641.21  1030.6 1709.45
#Mann= 3 , 0 , 0
       0      .1       0   466.3    .045       0   491.3     .08       0
Bank Sta=466.3,491.3
XS Rating Curve= 0 ,0
Exp/Cntr=0.3,0.1

Type RM Length L Ch R = 1 ,14068   ,203.6,174.2,144.8
XS GIS Cut Line= 4
     1777099.604      120912.082     1776998.288      121293.121
     1777048.946      121555.223     1777174.491      121914.237
#Sta/Elev= 30
    10.1 1670.26    20.2  1665.3    50.5 1648.63    60.7 1643.85    80.9 1635.69
   111.2 1625.09   121.3 1622.22   141.5  1617.9   192.1 1609.14   242.6 1599.08
   333.6 1578.02   384.2 1568.87   404.2 1562.35   414.1 1558.25   443.7 1545.42
   473.4 1531.03   480.7 1530.41   493.2 1530.11   505.7 1530.42   631.6 1538.18
   651.3 1540.67   701.3 1548.62   721.3 1553.29   771.3 1569.44   831.4 1592.09
   861.4  1604.7   921.5 1631.26   981.5 1655.44  1011.5 1668.96  1041.6 1683.69
#Mann= 3 , 0 , 0
    10.1     .08       0   480.7    .045       0   505.7     .08       0
#XS Ineff= 2 , 0
                           548.5         1541.14
Permanent Ineff=
       F       F
Bank Sta=480.7,505.7
XS Rating Curve= 0 ,0
Exp/Cntr=0.3,0.1

Type RM Length L Ch R = 1 ,13893.8 ,133.8,148.4,163
XS GIS Cut Line= 4
     1776718.363      121053.438     1776802.185      121442.612
      1776969.83      121502.485     1777135.478      121923.591
#Sta/Elev= 30
      10 1715.33    49.8 1692.47    99.5 1662.13   109.5 1654.85   139.3 1627.29
   149.3 1619.56   159.2 1614.05   169.2  1610.6     209 1602.72   308.5 1562.83
   368.2 1542.94   378.2 1540.85   398.1 1539.12   437.7 1538.74   447.5 1537.22
   464.7 1531.47   477.2 1530.07   489.7 1530.15   576.1 1534.88   606.3 1537.28
   666.6 1545.91     737 1558.51   787.3 1574.38   817.5    1585   897.9 1617.93
   938.1 1629.76   958.2 1636.72   998.5 1652.82  1008.5 1657.42  1028.6 1668.75
#Mann= 3 , 0 , 0
       0     .08       0   464.7    .045       0   489.7     .08       0
Bank Sta=464.7,489.7
XS Rating Curve= 0 ,0
Exp/Cntr=0.3,0.1

Type RM Length L Ch R = 1 ,13745.4 ,100.9,120.4,139.8
XS GIS Cut Line= 4
     1776628.554      121103.332     1776778.236      121540.405
     1776923.927      121708.049     1777073.609       121985.46
#Sta/Elev= 30
      10 1703.26    90.4 1659.81   180.8 1614.53     241 1586.16   261.1 1577.27
   281.2 1568.82   331.4 1549.76   351.5 1543.34   361.6 1541.16   371.6 1539.72
   411.8  1535.3   451.9 1531.59   520.2 1527.66   532.7 1527.09   542.8 1528.65
   545.2 1529.91   562.9 1539.61     573 1542.57   603.3 1545.35   613.4 1546.65
   653.8 1553.87   684.1 1561.21   733.3 1574.27   782.6 1585.44   802.3 1589.14
   861.4 1599.03   871.3 1601.44   881.1 1604.04   910.7 1614.05   999.3 1649.78
#Mann= 3 , 0 , 0
       0     .08       0   520.2    .045       0   545.2     .08       0
Bank Sta=520.2,545.2
XS Rating Curve= 0 ,0
Exp/Cntr=0.3,0.1

Type RM Length L Ch R = 1 ,13625.1 ,277.1,276.8,276.5
XS GIS Cut Line= 4
     1776520.097      121103.656     1776707.552      121374.615
     1776718.565      121740.236      1777056.27       122030.47
#Sta/Elev= 30
      10 1751.34    49.9 1733.28   139.8 1680.46   199.7 1649.45   299.5 1587.82
   329.5 1570.71   359.1 1561.04   398.7 1543.85   408.6 1541.31   497.5 1529.76
   564.1 1523.81   576.6 1522.93   589.1 1523.36   665.6 1540.31   695.3 1552.53
   715.1 1557.49   744.7 1567.62   784.3 1585.69   843.7 1616.05   863.5 1627.92
   883.3 1635.16     913 1639.84   922.9 1639.63   942.7 1635.12   952.5 1635.15
   992.1 1643.23  1031.7 1646.25  1110.9 1641.29  1130.7 1644.29  1140.6 1648.08
#Mann= 3 , 0 , 0
       0     .08       0   564.1    .045       0   589.1     .08       0
Bank Sta=564.1,589.1
XS Rating Curve= 0 ,0
Exp/Cntr=0.3,0.1

Type RM Length L Ch R = 1 ,13348.3 ,509.6,509,508.3
XS GIS Cut Line= 3
     1776420.409      121117.948     1776440.413      121618.049
     1776460.417      122118.149
#Sta/Elev= 30
      10 1733.62    90.1 1686.51   160.2 1642.47   210.2 1609.32   240.2 1590.34
   250.3 1583.45   280.3 1561.43   290.3 1555.88   300.3 1552.62   430.4 1525.42
   450.5 1523.34     488  1520.9   500.5 1520.63   510.5  1522.6   530.5 1533.77
   540.5 1538.77   590.6 1560.07   620.6 1573.96   640.6 1584.14   650.7 1590.32
   670.7 1605.15   740.7 1663.22   760.8 1679.05   860.9 1753.14   910.9 1788.29
   930.9 1801.27   940.9  1805.2     961 1807.41     971 1809.87    1001 1822.78
#Mann= 3 , 0 , 0
      10     .08       0     488    .045       0   510.5     .08       0
Bank Sta=488,510.5
XS Rating Curve= 0 ,0
Exp/Cntr=0.3,0.1

Type RM Length L Ch R = 1 ,12839.3 ,277.2,277.6,278.3
XS GIS Cut Line= 2
     1775903.753      121150.647     1775965.495      122123.083
#Sta/Elev= 30
      10 1702.47    20.1 1695.05    30.1 1686.48    50.2 1667.68    60.3 1659.77
    70.3 1653.19    90.4 1641.88   120.5 1627.04   140.6 1618.16   190.9 1599.07
     211 1590.36   361.6 1521.29   371.7 1517.56   381.7 1515.86     452  1515.6
   489.8 1514.38   502.3  1513.9   514.8 1514.44   522.4 1515.95   532.4 1521.12
   542.4  1527.8   622.8 1573.75   713.2 1622.03   743.4 1636.51   783.5 1653.81
   823.7    1668   853.9 1675.65   914.1 1684.83   954.3 1689.61   974.4 1691.12
#Mann= 3 , 0 , 0
      10     .06       0   489.8    .045       0   514.8     .06       0
#XS Ineff= 2 , 0
          412.64  1550.7
Permanent Ineff=
       F       F
Bank Sta=489.8,514.8
XS Rating Curve= 0 ,0
Exp/Cntr=0.3,0.1

Type RM Length L Ch R = 1 ,12561.7 ,369.3,369.6,369.5
XS GIS Cut Line= 3
     1775633.488      121175.692     1775662.147      121654.947
     1775679.795      122163.563
#Sta/Elev= 30
      10 1662.84      30 1651.28      40 1645.95      50 1641.21     120 1611.79
     140 1604.32     170 1593.96     190 1586.28     200 1582.06   280.1 1545.74
   340.1 1520.25   350.1 1516.26   360.1 1513.36   370.1 1511.99   410.1  1511.3
   460.1 1511.18   487.6  1510.1   500.1 1509.75   512.6 1510.44     530  1512.4
     540 1513.19   599.9  1515.7   629.8 1517.68   669.7  1521.2   739.6    1526
   779.5 1528.36   829.4 1530.61   879.3  1531.4   909.2 1532.49     989 1536.59
#Mann= 3 , 0 , 0
      10     .06       0   487.6    .045       0   512.6     .06       0
#XS Ineff= 2 , 0
          398.99 1534.33
Permanent Ineff=
       F       F
Bank Sta=487.6,512.6
XS Rating Curve= 0 ,0
Exp/Cntr=0.3,0.1

Type RM Length L Ch R = 1 ,12192.2 ,255.3,254.5,253.6
XS GIS Cut Line= 2
     1775276.043      121176.373     1775317.204      122159.099
#Sta/Elev= 30
      10 1671.45    50.2  1650.3   120.4 1609.27   160.6 1588.81   220.8 1552.92
   250.9 1539.44     271 1534.59     281 1533.44   301.1 1534.31   311.1 1531.92
   341.2 1513.57   351.3 1508.93   361.3 1506.78   421.5  1505.5   469.3 1500.31
   481.8 1500.02   494.3 1501.05   592.2 1510.73   622.3 1516.52   652.4 1529.01
   722.6 1570.15   782.9    1596     813  1604.5   843.1  1609.8   883.2 1614.87
   923.4  1615.5   943.4 1617.89   953.5 1621.71   973.6 1633.45   983.6 1637.36
#Mann= 3 , 0 , 0
       0     .06       0   469.3    .045       0   494.3     .06       0
Bank Sta=469.3,494.3
XS Rating Curve= 0 ,0
Exp/Cntr=0.3,0.1

Type RM Length L Ch R = 1 ,11937.7 ,285.9,286.4,287
XS GIS Cut Line= 3
     1775006.077      121177.305     1775043.054      121676.437
     1775080.032      122175.569
#Sta/Elev= 30
      10 1679.07    70.1  1640.5    80.1 1633.39   110.1  1609.7   130.1 1596.42
   160.2 1578.63   210.2 1551.27   260.3 1519.61   280.3 1508.64   290.3 1505.23
   300.3 1503.65   350.4 1504.11   420.4 1502.37     468 1497.95   480.5 1497.12
     493  1498.7   540.5 1509.43   550.6 1513.04   560.6 1518.67   580.6 1532.83
   620.6 1563.78   640.6 1577.65   680.7 1603.72   730.7 1637.55   850.9 1714.12
     961 1786.53     971 1791.99     981 1795.73     991 1797.59    1001 1798.29
#Mann= 3 , 0 , 0
       0     .06       0     468    .045       0     493     .06       0
Bank Sta=468,493
XS Rating Curve= 0 ,0
Exp/Cntr=0.3,0.1

Type RM Length L Ch R = 1 ,11651.3 ,313,310.6,308.7
XS GIS Cut Line= 2
     1774730.656      121202.098     1774782.107      122164.244
#Sta/Elev= 30
      10 1606.71    40.1 1601.07    60.2 1599.36    70.3 1597.26    80.3  1593.3
   140.5 1559.83   160.6 1549.27   230.8 1517.01   240.9 1513.36     271 1506.43
   311.1 1499.96   411.5 1497.93   421.5 1497.33   449.2 1494.08   461.7 1492.84
   471.7 1492.93   474.2 1493.52   481.8 1495.29   501.8 1505.54   511.9 1510.15
   562.1 1531.63   592.2 1545.56   712.6 1608.47   732.7 1620.65   752.8 1634.48
   792.9 1663.78   843.1 1701.96   883.2 1730.37   923.4  1757.2   963.5 1780.42
#Mann= 3 , 0 , 0
       0     .06       0   449.2    .045       0   474.2     .06       0
Bank Sta=449.2,474.2
XS Rating Curve= 0 ,0
Exp/Cntr=0.3,0.1

Type RM Length L Ch R = 1 ,11340.7 ,601.1,599.6,597.6
XS GIS Cut Line= 3
     1774365.349      121135.211     1774452.457      121720.479
     1774514.559       122189.97
#Sta/Elev= 30
      10 1602.23    50.1 1597.27    70.2 1592.29    90.3 1584.26   120.3 1570.63
   140.4  1564.5   160.5 1561.77   190.6 1564.52   230.7 1561.49   240.7 1558.81
   270.8 1544.23   290.8 1532.81     331 1507.75     341 1502.38     351 1498.53
     361 1496.94   411.2 1496.25   569.2 1489.85   581.7 1489.33   594.2 1490.63
   601.8 1493.02   611.9 1498.43   692.5  1543.5   813.4 1616.58   873.8 1651.37
     894 1665.19   934.3 1696.59  1004.8 1746.61    1025 1759.29  1065.3 1779.24
#Mann= 3 , 0 , 0
       0     .06       0   569.2    .045       0   594.2     .06       0
Bank Sta=569.2,594.2
XS Rating Curve= 0 ,0
Exp/Cntr=0.3,0.1

Type RM Length L Ch R = 1 ,10741   ,688.1,683.8,680
XS GIS Cut Line= 3
     1773762.214      121309.236     1773860.364      121799.993
     1773961.081      122290.396
#Sta/Elev= 30
      10 1696.01      30 1680.03    70.1 1645.23   100.1  1620.3   120.1 1604.98
   150.1 1583.37   190.2 1555.73   220.2 1536.46   250.2 1519.93   290.3 1500.31
   310.3 1492.93   320.3 1490.93   370.4 1484.58     478 1481.98   490.5 1481.52
   500.5 1482.06     503 1482.86   510.5 1485.25   540.5 1502.58   590.6 1528.71
   650.7 1565.62   700.7 1594.04   720.8 1604.56   770.8  1628.8   810.9 1650.73
   830.9 1663.43     881 1702.29     891 1709.28     901 1715.11  1001.1 1757.33
#Mann= 3 , 0 , 0
       0     .06       0     478    .045       0     503     .06       0
Bank Sta=478,503
XS Rating Curve= 0 ,0
Exp/Cntr=0.3,0.1

Type RM Length L Ch R = 1 ,10057.2 ,493.8,489.6,485.1
XS GIS Cut Line= 3
     1773037.641      121535.221      1773210.87      122004.865
     1773376.775      122477.054
#Sta/Elev= 30
      10 1646.07    90.1 1599.31   160.2 1556.81   210.2 1524.03   220.3 1516.82
   250.3 1493.12   260.3 1486.03   270.3  1480.5   280.3 1477.47   290.3 1476.71
   340.4 1476.74   460.5 1474.89   470.5 1474.65   488.1 1472.67   500.6 1471.35
   510.6 1472.71   513.1 1474.02   520.6 1477.96   540.6 1491.46   610.7 1529.52
   750.8 1611.67   780.8 1632.08   850.9 1684.51   880.9 1705.96     911  1725.9
     921 1731.84     951 1746.75     961 1753.24   991.1 1776.95  1001.1 1784.05
#Mann= 3 , 0 , 0
      10     .06       0   488.1    .045       0   513.1     .06       0
#XS Ineff= 2 , 0
          430.34 1494.96
Permanent Ineff=
       F       F
Bank Sta=488.1,513.1
XS Rating Curve= 0 ,0
Exp/Cntr=0.3,0.1

Type RM Length L Ch R = 1 ,9567.7  ,285.9,298.6,326.6
XS GIS Cut Line= 3
       1772498.5      121724.819     1772784.673      122239.802
     1773016.097      122660.898
#Sta/Elev= 30
      10 1679.17    99.9 1626.47   119.8 1614.08   159.8 1583.84   229.7 1533.12
   249.6 1519.59   269.6  1508.4   299.6 1495.13   309.6 1491.44   319.5 1489.09
   389.4 1474.22   419.4 1469.28   439.4 1467.61   479.3 1467.45   566.7 1465.06
   579.2    1465   591.7 1465.37   599.2 1466.36   639.2 1485.31   659.2  1495.4
   669.2 1501.27   739.3 1545.59   759.3 1556.34   809.4 1580.87   869.4 1602.25
   919.5 1622.14   949.5 1631.93   959.5 1634.54  1019.6  1645.9  1069.7 1653.23
#Mann= 3 , 0 , 0
      10     .06       0   566.7    .045       0   591.7     .06       0
#XS Ineff= 2 , 0
          493.82 1491.97
Permanent Ineff=
       F       F
Bank Sta=566.7,591.7
XS Rating Curve= 0 ,0
Exp/Cntr=0.3,0.1

Type RM Length L Ch R = 1 ,9269.1  ,346.3,328.1,308.9
XS GIS Cut Line= 4
     1772420.477      121696.034     1772593.209      122030.971
     1772461.638      122323.744      1772513.09      122699.341
#Sta/Elev= 30
     9.9 1724.92    29.8 1709.08    39.7 1702.24    59.5 1691.64     119 1657.36
   168.6 1627.52   178.5 1621.91   208.3 1607.09   228.1  1594.7   247.9 1580.29
   327.3 1517.44   347.1 1502.53     357 1496.05   366.9 1491.31   376.9    1488
     417 1478.22   457.1  1465.9   467.1 1463.87   494.8 1460.85   507.3 1459.92
   519.8 1460.25   527.3 1461.12   547.4 1465.91   557.4 1466.74   707.8 1468.55
   797.6 1468.15   917.3 1473.12   947.2 1477.69    1037 1499.16  1076.9 1507.71
#Mann= 3 , 0 , 0
       0     .06       0   494.8    .045       0   519.8     .06       0
Bank Sta=494.8,519.8
XS Rating Curve= 0 ,0
Exp/Cntr=0.3,0.1

Type RM Length L Ch R = 1 ,8941    ,589.9,600,611.5
XS GIS Cut Line= 3
     1772119.754      121739.271      1772227.25      122231.182
     1772350.722      122716.798
#Sta/Elev= 30
    10.1 1658.16    30.2 1636.64    40.3 1627.23    60.4 1610.35    90.6 1589.35
   110.8 1576.82   130.9 1565.93   151.1 1556.46   171.2 1548.56   191.3  1542.3
     282 1522.02   332.3 1509.11   372.6 1493.41   443.1 1468.23   463.2 1462.05
     491 1456.73   503.5 1455.42     516 1455.57   593.7 1461.46   683.9 1463.81
   693.9 1464.71   703.9 1467.19     714  1471.6     724 1477.28   854.3 1553.79
   874.3  1564.4   884.3 1568.73   894.4 1572.21   924.4 1579.94  1004.6 1597.13
#Mann= 3 , 0 , 0
       0     .06       0     491    .045       0     516     .06       0
Bank Sta=491,516
XS Rating Curve= 0 ,0
Exp/Cntr=0.3,0.1

Type RM Length L Ch R = 1 ,8341    ,599.8,600,601.5
XS GIS Cut Line= 3
      1771717.04      121717.701     1771643.411      122213.564
      1771561.93       122707.09
#Sta/Elev= 30
      10 1672.82    20.1 1665.62    30.1  1659.3    90.2  1624.8   120.3 1609.14
   170.4 1584.81   210.5 1567.12   260.7 1546.18   280.7  1538.5   330.9 1520.84
     381 1501.34   461.2 1466.58   481.2 1455.57   488.8 1452.53   491.3 1451.53
   501.3 1450.36   513.8  1451.1   541.3 1453.22   611.3 1455.83   621.3 1457.78
   631.4 1462.63   701.4 1504.76   841.4 1592.04   871.5  1612.3   911.5 1640.42
   951.5 1667.64   961.5 1674.04   971.5 1679.35   981.5 1682.99  1001.5 1687.16
#Mann= 3 , 0 , 0
       0     .06       0   488.8    .045       0   513.8     .06       0
Bank Sta=488.8,513.8
XS Rating Curve= 0 ,0
Exp/Cntr=0.3,0.1

Type RM Length L Ch R = 1 ,7741    ,211.3,205,196.8
XS GIS Cut Line= 3
     1771128.117      121662.502      1771050.25      122159.926
     1770941.806      122647.922
#Sta/Elev= 30
    10.1 1573.47    40.3 1559.26    60.4 1551.07    90.6 1537.23   120.8 1524.91
   161.1 1511.04   201.4 1498.67   241.7  1488.4   322.2 1470.31   372.6 1456.03
   382.6 1453.58   402.8 1450.75   480.9 1442.12   493.4 1441.91   505.9 1443.53
   523.5 1446.96   593.5 1454.79   663.4 1458.12   673.4 1459.93   683.4 1462.52
   693.4 1465.72   703.4 1469.79   723.4 1480.35   763.4 1503.71   803.4 1526.35
   873.4 1567.98   893.4 1581.24   963.4 1630.97   983.4 1646.11  1003.4 1659.97
#Mann= 3 , 0 , 0
       0     .06       0   480.9    .045       0   505.9     .06       0
Bank Sta=480.9,505.9
XS Rating Curve= 0 ,0
Exp/Cntr=0.3,0.1

Type RM Length L Ch R = 1 ,7536.1  ,207.5,223.4,239.3
XS GIS Cut Line= 4
     1771013.989      121627.907     1770846.595      122017.756
     1770859.811      122213.782      1770824.57      122552.973
#Sta/Elev= 30
    10.1 1631.37    30.3 1627.87    50.5    1626    60.6 1622.53    70.7 1617.05
    90.9 1604.56     101 1597.44   121.2 1581.57   161.6 1547.47   181.8 1532.26
   212.1 1510.82   232.3 1497.56   252.5 1485.72   272.7 1475.58   292.9 1466.98
   323.3  1456.8   343.5 1452.29   434.1 1448.23   500.2 1441.14   512.7  1440.3
   525.2 1440.92   561.8 1445.08     711 1454.87     721 1457.29   731.1 1461.71
   771.2  1483.1   811.3 1506.81   851.4 1528.79   911.6  1564.2   961.8 1595.67
#Mann= 3 , 0 , 0
       0     .08       0   500.2    .045       0   525.2     .08       0
Bank Sta=500.2,525.2
XS Rating Curve= 0 ,0
Exp/Cntr=0.3,0.1

Type RM Length L Ch R = 1 ,7312.7  ,171.9,171.6,171.4
XS GIS Cut Line= 4
     1770853.203      121568.438     1770692.418      121945.072
     1770580.088      122149.909     1770443.531      122436.239
#Sta/Elev= 30
      10 1728.91      30 1726.04    59.9 1714.46    89.9  1697.9   109.9  1682.9
   129.8 1663.01   149.8 1639.05   169.8  1611.4   219.7 1534.93   229.7 1522.93
   239.7  1513.1   259.7 1499.42   289.7 1485.52   319.6 1476.28   389.5 1461.34
   477.7 1445.36   513.8 1436.73   526.3 1435.73   538.8 1439.36   584.7 1447.02
   633.4 1450.51   672.9 1450.58   742.3  1447.2     772 1448.78   791.8  1454.4
   821.6 1473.23   851.3  1486.5   900.9 1502.11   940.5 1511.68   960.4 1520.61
#Mann= 3 , 0 , 0
       0     .06       0   513.8    .045       0   538.8     .06       0
Bank Sta=513.8,538.8
XS Rating Curve= 0 ,0
Exp/Cntr=0.3,0.1

Type RM Length L Ch R = 1 ,7141    ,562.3,571.7,580.2
XS GIS Cut Line= 3
     1770724.139      121520.863     1770487.548      121961.913
     1770250.958      122402.963
#Sta/Elev= 30
      10 1766.44      40 1746.86      50 1737.45    60.1 1725.17    80.1 1697.75
    90.1 1685.65   100.1 1674.81   120.1 1655.97   150.2 1630.68   190.2 1601.24
   230.2 1575.87   270.3 1553.09   420.4 1481.66   440.4 1470.71   490.5 1440.08
     498 1436.63   500.5 1435.48   510.5 1434.64     523 1437.93   530.5 1440.09
   540.5 1441.04   700.7 1440.84   720.7 1442.29   730.7 1446.36   750.8 1457.38
   810.8 1493.43   850.8 1512.62   870.9 1523.83   930.9 1558.64    1001 1601.28
#Mann= 3 , 0 , 0
       0     .06       0     498    .045       0     523     .06       0
Bank Sta=498,523
XS Rating Curve= 0 ,0
Exp/Cntr=0.3,0.1

Type RM Length L Ch R = 1 ,6569.3  ,311.9,309.6,308.4
XS GIS Cut Line= 3
     1770417.219      121295.234     1770025.796      121639.379
      1769681.46      121974.395
#Sta/Elev= 30
      10  1612.4      20 1608.01   100.2 1576.17   140.3 1558.17   210.5 1524.64
   220.5 1520.38   240.6 1513.92   250.6 1510.95   260.6  1508.9   300.7 1504.46
   380.9 1493.04   400.9  1489.2     431 1481.57     451 1478.56   461.1 1476.08
   471.1 1469.66   481.1 1460.36   491.1 1448.94   501.2 1435.47   511.2 1425.42
   521.2 1421.93   533.7 1422.56   601.3 1430.58   691.3 1435.13   711.4 1435.65
   811.5 1434.13   841.5  1435.1   871.5 1438.17   971.6 1452.29  1001.6 1455.68
#Mann= 3 , 0 , 0
      10     .08       0   511.2    .045       0   533.7     .08       0
Bank Sta=511.2,533.7
XS Rating Curve= 0 ,0
Exp/Cntr=0.3,0.1

Type RM Length L Ch R = 1 ,6259.7  ,321.1,318.7,316.2
XS GIS Cut Line= 2
     1770146.314      121063.179     1769477.443      121778.357
#Sta/Elev= 30
    10.1 1688.53    40.4 1683.74    60.6 1679.73    80.8 1674.65     101 1667.93
   121.1 1659.54   151.4 1644.84   201.9 1617.79   232.2  1600.5   292.8 1561.25
   312.9 1546.73     424  1452.5   434.1 1443.37   454.3 1423.18     462 1419.64
   464.4 1418.53   474.5 1418.34     487 1418.95   615.8 1423.84   656.2 1430.75
   676.4 1432.45     747 1432.22   827.8 1433.67   837.9 1435.42   858.1 1443.89
   868.2 1447.35   888.4 1453.24   908.6 1458.02   938.8 1462.85   979.2 1466.38
#Mann= 3 , 0 , 0
    10.1     .06       0     462    .045       0     487     .06       0
#XS Ineff= 2 , 0
                          573.57         1476.06
Permanent Ineff=
       F       F
Bank Sta=462,487
XS Rating Curve= 0 ,0
Exp/Cntr=0.3,0.1

Type RM Length L Ch R = 1 ,5941    ,437,444.8,451.7
XS GIS Cut Line= 3
      1769869.28      120831.914     1769561.761      121226.796
     1769254.241      121621.679
#Sta/Elev= 30
      10 1677.03      50 1652.28   160.2  1589.6   230.2 1548.34   250.2 1535.28
   270.3 1520.97   280.3  1515.9   290.3 1513.14   320.3 1511.36   330.3 1508.28
   460.5 1434.11     488 1416.83   500.5 1411.95     513 1412.77   540.5  1418.8
   600.6 1418.97   620.6 1420.26   740.7 1440.24   770.8 1443.66   780.8  1446.6
   830.8 1469.14   840.8 1474.66   850.8  1482.8   880.9 1514.88   890.9 1524.73
   900.9 1532.16   910.9 1537.79   950.9 1556.59     971 1562.09    1001 1568.04
#Mann= 3 , 0 , 0
       0     .08       0     488    .045       0     513     .08       0
Bank Sta=488,513
XS Rating Curve= 0 ,0
Exp/Cntr=0.3,0.1

Type RM Length L Ch R = 1 ,5496.2  ,415.3,417.9,421.3
XS GIS Cut Line= 3
     1769667.814      120610.405     1769248.606      120913.049
     1768880.604      121196.953
#Sta/Elev= 30
     9.9 1665.69    79.5 1623.95   119.3 1604.64   228.7 1549.42   377.8 1475.92
   457.4 1437.42   487.2 1421.48   507.1  1408.7   514.6 1405.11     517 1403.96
   527.1 1403.25   539.6 1405.88   557.5 1410.37   567.6 1411.02   638.3  1408.7
   658.5 1409.24   668.6 1411.62   719.1 1432.48   729.2 1435.91   749.4 1439.19
   759.5 1442.17   769.6  1446.5     800 1460.05   810.1 1465.22   820.2 1472.74
   830.3 1483.02   850.5 1506.15   860.6  1516.8   870.7 1524.93   981.8 1596.64
#Mann= 3 , 0 , 0
     9.9     .06       0   514.6    .045       0   539.6     .06       0
#XS Ineff= 2 , 0
                           575.6         1448.46
Permanent Ineff=
       F       F
Bank Sta=514.6,539.6
XS Rating Curve= 0 ,0
Exp/Cntr=0.3,0.1

Type RM Length L Ch R = 1 ,5078.4  ,722.8,731.3,739.8
XS GIS Cut Line= 3
     1769463.455      120304.662     1769031.866       120557.51
     1768602.765      120811.066
#Sta/Elev= 30
      10 1727.89      50 1702.48      80 1681.96     100 1667.35     120 1651.16
   150.1  1625.2   190.1 1593.42   260.1 1535.07   280.1 1520.08   330.1 1484.97
   360.1 1467.39   390.2 1451.76   430.2 1433.03   490.2 1406.37   510.2 1395.81
   517.6 1393.35   520.1 1392.51   530.1 1392.03   542.6 1392.46   679.6 1397.97
   709.5 1401.32   729.5 1405.62   739.4 1408.96   769.3 1422.39   779.3 1425.31
   799.3 1429.62   809.2 1435.51   829.2 1449.53   938.8 1529.85   998.6 1572.59
#Mann= 3 , 0 , 0
      10     .06       0   517.6    .045       0   542.6     .06       0
#XS Ineff= 2 , 0
                          610.19         1559.59
Permanent Ineff=
       F       F
Bank Sta=517.6,542.6
XS Rating Curve= 0 ,0
Exp/Cntr=0.3,0.1

Type RM Length L Ch R = 1 ,4347.1  ,961.8,960.4,959
XS GIS Cut Line= 4
     1769174.724      119771.493     1768973.217      119864.356
     1768520.442      119972.404     1768206.587      120085.598
#Sta/Elev= 30
    10.1 1673.49    50.4 1674.77    60.5 1670.41    70.6 1661.57    90.8 1638.22
   110.9 1622.23   141.2  1603.5   181.5  1580.4   251.6 1534.93   281.3 1516.89
   291.2 1509.94   320.9  1483.7   340.7 1470.66     420 1421.45   449.7 1405.72
   469.5 1397.35   516.4 1386.68   528.9  1384.6   541.4 1384.91   568.5 1387.78
   637.8 1389.26   667.6 1391.63   697.5 1396.24   758.1 1397.17   768.2 1398.82
   778.4 1403.85   828.9 1440.06   899.7 1488.28   960.3 1538.51    1021 1583.09
#Mann= 3 , 0 , 0
    10.1     .08       0   516.4    .045       0   541.4     .06       0
#XS Ineff= 2 , 0
                          594.65         1525.65
Permanent Ineff=
       F       F
Bank Sta=516.4,541.4
XS Rating Curve= 0 ,0
Exp/Cntr=0.3,0.1

Type RM Length L Ch R = 1 ,3386.7  ,319,310.1,301.2
XS GIS Cut Line= 3
     1769023.744      118853.208     1768543.628      118994.262
      1768063.67      119136.704
#Sta/Elev= 30
      10  1650.6   130.1 1566.88   190.2 1530.33   220.2 1511.08   250.2 1493.76
   380.3 1430.02   390.3 1425.83   400.3  1422.9   440.4 1414.05   450.4 1409.92
   510.4 1380.67   530.4 1369.58     538 1367.32   550.5 1366.44     563 1368.56
   580.5 1371.31   600.5 1372.09   610.6 1373.48   640.6    1381   660.6 1381.73
   670.6 1384.67   680.6 1391.04   710.7 1412.67   750.7 1439.18   760.7 1444.58
   780.8 1452.16   810.8 1459.11     921 1475.09     961 1484.97  1001.1 1496.19
#Mann= 3 , 0 , 0
      10     .08       0     538    .045       0     563     .08       0
#XS Ineff= 2 , 0
                          576.27         1401.98
Permanent Ineff=
       F       F
Bank Sta=538,563
XS Rating Curve= 0 ,0
Exp/Cntr=0.3,0.1

Type RM Length L Ch R = 1 ,3076.6  ,749,749.5,749.7
XS GIS Cut Line= 3
     1768850.091      118416.621     1768242.962      118828.234
     1767990.849      119003.169
#Sta/Elev= 30
      10  1599.3    30.1 1589.77   170.8  1540.2     201 1528.56   221.1 1519.36
   251.2 1504.06   291.4 1487.69   331.6 1469.73   351.7 1459.42   391.9 1435.71
   432.1 1414.54   482.3 1384.42   502.4 1370.41   512.4 1364.15     520 1361.77
   522.5 1360.99   532.5 1360.91     545 1362.11   582.8 1365.82   703.4 1371.54
   743.4 1377.51   753.3 1380.23   773.1 1387.95   792.9 1396.24   842.4 1421.76
     882  1443.3   921.6 1466.29   931.5 1472.85   971.1  1505.3  1040.4 1555.83
#Mann= 3 , 0 , 0
       0     .08       0     520    .045       0     545     .08       0
Bank Sta=520,545
XS Rating Curve= 0 ,0
Exp/Cntr=0.3,0.1

Type RM Length L Ch R = 1 ,2327.1  ,300,291.1,282.5
XS GIS Cut Line= 3
     1768385.461      117876.522     1767962.126      118142.277
     1767539.615      118431.684
#Sta/Elev= 30
      10 1659.32   159.9 1563.56   249.9  1509.4   279.9 1490.73   309.9 1470.84
   359.9 1436.14   369.9 1428.83   399.9 1405.12   409.9 1398.18   419.9 1392.32
   429.9 1388.25   449.9 1384.17   459.9 1381.15   469.8 1376.85   489.8 1366.21
   509.9 1353.77   519.9 1350.56   537.5 1350.12     550  1350.1   562.5 1350.11
   620.3 1351.83   650.5 1355.85   690.6  1360.2   700.7 1364.41   710.7 1371.38
   720.8 1379.57   861.3 1496.93   911.5 1538.12   951.7 1570.44    1012 1617.79
#Mann= 3 , 0 , 0
       0     .06       0   537.5    .045       0   562.5     .06       0
Bank Sta=537.5,562.5
XS Rating Curve= 0 ,0
Exp/Cntr=0.3,0.1

Type RM Length L Ch R = 1 ,2036    ,638.3,627.1,616.1
XS GIS Cut Line= 5
     1767993.143      117352.489     1767968.416      117566.208
     1767915.555      117729.196     1767635.832      118083.805
     1767535.224      118432.973
#Sta/Elev= 30
     9.8 1511.95      88 1470.78     176 1443.36   205.4 1436.97   245.4 1433.82
   285.7  1426.5   336.1 1425.14   376.4 1421.17   426.6 1411.43   476.8 1405.02
   486.9 1402.82   496.9 1398.68     537 1376.54   567.2 1364.47   597.3 1358.03
   627.4  1355.1   665.1 1345.69   677.6  1345.2   690.1 1347.43   707.7 1350.27
   767.9 1348.22     798 1348.86     808 1350.29   818.1 1354.42   888.6  1406.7
   959.3  1463.6   989.6 1486.02  1029.9  1512.6    1141 1581.65  1201.5 1621.02
#Mann= 3 , 0 , 0
       0     .06       0   665.1    .045       0   690.1     .06       0
Bank Sta=665.1,690.1
XS Rating Curve= 0 ,0
Exp/Cntr=0.3,0.1

Type RM Length L Ch R = 1 ,1408.9  ,601.7,584.6,567.4
XS GIS Cut Line= 3
     1767311.329      117204.306     1767184.528      117687.156
      1767043.78      118212.758
#Sta/Elev= 30
      10 1573.11   119.8 1508.78   139.8  1496.4   219.7 1442.21   289.5 1391.79
   299.5 1387.95   329.5 1385.53   339.5 1381.98   349.5 1376.22   369.4 1362.29
   389.4 1347.07   399.4 1341.08   409.4 1338.05   486.7 1331.23   499.2 1330.91
   511.7 1333.27   519.4 1335.11   529.5 1335.75   559.7  1335.3   579.8 1336.53
   620.1 1341.23   630.2 1343.31   640.3 1346.54   690.7 1365.94   710.8 1374.75
   811.6 1424.91   821.7 1429.09   922.4 1465.46  1023.2 1496.34  1043.3 1503.48
#Mann= 3 , 0 , 0
       0     .08       0   486.7    .045       0   511.7     .08       0
Bank Sta=486.7,511.7
XS Rating Curve= 0 ,0
Exp/Cntr=0.3,0.1

Type RM Length L Ch R = 1 ,824.2   ,207.7,226.2,244.6
XS GIS Cut Line= 4
     1766512.889      117192.912     1766549.844       117507.87
     1766683.619      117862.887     1766601.296       118264.21
#Sta/Elev= 30
     9.9 1492.89    69.4  1511.2    79.3 1513.33    89.2 1512.55    99.1 1507.84
   118.9 1491.03   178.4 1431.11   188.3 1422.56   198.2 1417.27     218 1411.95
   227.9  1406.3   297.3 1347.26   307.2 1339.85   317.1 1334.14   327.1  1331.1
     387 1327.34   466.9 1324.27   556.7 1326.94   574.2 1323.65   586.7 1323.06
   596.7 1326.49   616.6 1340.78   636.6 1352.15   706.5 1388.52   746.5 1410.63
   766.4 1420.26   826.4 1441.72   946.3  1477.4  1016.3 1500.55  1106.2  1534.8
#Mann= 3 , 0 , 0
     9.9     .06       0   574.2    .045       0   596.7     .06       0
Bank Sta=574.2,596.7
XS Rating Curve= 0 ,0
Exp/Cntr=0.3,0.1

Type RM Length L Ch R = 1 ,598.1   ,300.6,313.1,325.5
XS GIS Cut Line= 4
     1766426.206      117177.664     1766464.126      117606.753
     1766364.151      117920.213     1766223.823      118179.038
#Sta/Elev= 30
      10 1420.26   130.2  1445.5   150.3 1447.48   160.3 1445.92   170.3 1441.29
   190.3 1425.85   200.4 1420.74   220.4 1415.79   230.4 1410.72   260.5 1386.16
   300.5  1346.2   310.5 1337.34   320.6 1331.37   330.6 1328.69   340.6 1327.79
   470.6 1318.28   500.6 1318.08   540.4 1321.31   557.8 1320.15   570.3 1317.09
   582.8 1318.03   590.3 1320.71   640.1 1349.05     690 1375.25   769.6 1423.21
   838.3  1469.8     907 1520.38   975.7 1567.87  1014.9 1591.77  1054.2 1612.29
#Mann= 3 , 0 , 0
      10     .06       0   557.8    .045       0   582.8     .06       0
#XS Ineff= 2 , 0
          499.43 1341.91
Permanent Ineff=
       F       F
Bank Sta=557.8,582.8
XS Rating Curve= 0 ,0
Exp/Cntr=0.3,0.1

Type RM Length L Ch R = 1 ,285     ,272.5,285,297.5
XS GIS Cut Line= 4
     1766420.219      117153.715     1766262.554      117487.007
     1766025.058      117744.461     1766039.839      118163.447
#Sta/Elev= 30
      10  1414.4    29.9 1414.63    49.8 1412.47    59.8 1410.15    79.7 1402.93
   109.6 1387.42   189.3 1341.28   199.3 1336.54   219.2 1329.12   249.1 1326.72
   388.7 1322.92   448.8 1318.63   488.8 1312.13   518.8 1310.92   536.3 1309.11
   548.8  1308.4   561.3 1308.73   598.9 1314.05   658.9 1318.55     719 1321.18
   758.9 1331.28   798.8 1333.69   808.8  1335.9   818.8 1340.77   838.8 1355.55
  1008.4 1502.47  1028.4 1518.38  1078.3 1554.01  1098.3 1565.68  1138.2 1585.82
#Mann= 3 , 0 , 0
      10     .06       0   536.3    .045       0   561.3     .06       0
#XS Ineff= 2 , 0
          508.13  1334.2
Permanent Ineff=
       F       F
Bank Sta=536.3,561.3
XS Rating Curve= 0 ,0
Exp/Cntr=0.3,0.1

Chan Stop Cuts=-1
Use User Specified Reach Order=0
